--- RENICKCK.prj (project) ---

Proj Title=RENICKCK
Current Plan=p01
Default Exp/Contr=0.3,0.1
English Units
Geom File=g01
Flow File=f01
Plan File=p01
Y Axis Title=Elevation
X Axis Title(PF)=Main Channel Distance
X Axis Title(XS)=Station
BEGIN DESCRIPTION:
Stream Name- Renick Creek
Flood Zone: Zone A
Greenbrier County, WV
County-Wide Study
WVDHSEM-2018-3, Flood Risk Project
HEC-RAS Version: 5.0.7
General Notes:
For the Hydrology Regression was used.
END DESCRIPTION:
DSS Export Rating Curves= 0
DSS Export Rating Curve Sorted= 0
DSS Export Volume Flow Curves= 0
DXF Filename=..\J2.
DXF OffsetX= 0
DXF OffsetY= 0
DXF ScaleX= 1
DXF ScaleY= 10

--- RENICKCK.p01 (plan) ---

Plan Title=Floodplain
Program Version=5.07
Short Identifier=Floodplain
Geom File=g01
Flow File=f01
Subcritical Flow
K Sum by GR= 0
Std Step Tol= 0.01
Critical Tol= 0.01
Num of Std Step Trials= 20
Max Error Tol= 0.3
Flow Tol Ratio= 0.001
Split Flow NTrial= 30
Split Flow Tol= 0.02
Split Flow Ratio= 0.02
Log Output Level= 0
Friction Slope Method= 1
Unsteady Friction Slope Method= 2
Unsteady Bridges Friction Slope Method= 1
Parabolic Critical Depth
Global Vel Dist= 0 , 0 , 0
Global Log Level= 0
CheckData=True
Encroach Param=-1 ,0,0, 0
Computation Interval=1MIN
Output Interval=1HOUR
Instantaneous Interval=1HOUR
Mapping Interval=1HOUR
Computation Time Step Use Courant=        0
Computation Time Step Use Time Series=    0
Computation Time Step Count To Double=0
Computation Time Step Max Doubling=0
Computation Time Step Max Halving=0
Computation Time Step Residence Courant=0
Run HTab= 0
Run UNet= 0
Run Sediment= 0
Run PostProcess= 0
Run WQNet= 0
Run RASMapper= 0
UNET Theta= 1
UNET Theta Warmup= 1
UNET ZTol= 0.02
UNET ZSATol= 0.02
UNET MxIter= 20
UNET Max Iter WO Improvement= 0
UNET MaxInSteps= 0
UNET DtIC= 0
UNET DtMin= 0
UNET MaxCRTS= 20
UNET WFStab= 2
UNET SFStab= 1
UNET WFX= 1
UNET SFX= 1
UNET 1D Methodology=Finite Difference
UNET DSS MLevel= 4
UNET Pardiso=0
UNET DZMax Abort= 100
UNET Use Existing IB Tables=-1
UNET Froude Reduction=False
UNET Froude Limit= 0.8
UNET Froude Power= 4
UNET D1 Cores= 0
UNET D2 Coriolis=0
UNET D2 Cores= 0
UNET D2 Theta= 1
UNET D2 Theta Warmup= 1
UNET D2 Z Tol= 0.01
UNET D2 Volume Tol= 0.01
UNET D2 Max Iterations= 20
UNET D2 Equation= 0
UNET D2 RampUpFraction=0.1
UNET D2 TimeSlices= 1
UNET D2 BCVolumeCheck=0
UNET D1D2 MaxIter= 0
UNET D1D2 ZTol=0.01
UNET D1D2 QTol=0.1
UNET D1D2 MinQTol=1
Write IC File= 0
Write IC File at Fixed DateTime=0
Write IC File at Sim End=0
Echo Input=False
Echo Parameters=False
Echo Output=False
Write Detailed= 0
HDF Write Warmup=0
HDF Write Time Slices=0
HDF Flush=0
HDF Face Node Velocities=0
HDF Compression= 1
HDF Chunk Size= 1
HDF Spatial Parts= 1
HDF Use Max Rows=0
HDF Fixed Rows= 1
Calibration Method= 0
Calibration Iterations= 20
Calibration Max Change=0.05
Calibration Tolerance=0.2
Calibration Maximum=1.5
Calibration Minimum=0.5
Calibration Optimization Method= 1
WQ AD Non Conservative
WQ ULTIMATE=-1
WQ Max Comp Step=1HOUR
WQ Output Interval=15MIN
WQ Output Selected Increments= 0
WQ Output face flow=0
WQ Output face velocity=0
WQ Output face area=0
WQ Output face dispersion=0
WQ Output cell volume=0
WQ Output cell surface area=0
WQ Output cell continuity=0
WQ Output cumulative cell continuity=0
WQ Output face conc=0
WQ Output face dconc_dx=0
WQ Output face courant=0
WQ Output face peclet=0
WQ Output face adv mass=0
WQ Output face disp mass=0
WQ Output cell mass=0
WQ Output cell source sink temp=0
WQ Output nsm pathways=0
WQ Output nsm derived pathways=0
WQ Output MaxMinRange=-1
WQ Daily Max Min Mean=-1
WQ Daily Range=0
WQ Daily Time=0
WQ Create Restart=0
WQ Fixed Restart=0
WQ System Summary=0
WQ Write To DSS=0
WQ Use Fixed Temperature=0
Sorting and Armoring Iterations= 10
XS Update Threshold= 0.02
Bed Roughness Predictor= 0
Hydraulics Update Threshold= 0.02
Energy Slope Method= 1
Volume Change Method= 1
Sediment Retention Method= 0
XS Weighting Method= 0
Number of US Weighted Cross Sections= 1
Number of DS Weighted Cross Sections= 1
Upstream XS Weight=0
Main XS Weight=1
Downstream XS Weight=0
Number of DS XS's Weighted with US Boundary= 1
Upstream Boundary Weight= 1
Weight of XSs Associated with US Boundary= 0
Number of US XS's Weighted with DS Boundary= 1
Downstream Boundary Weight= 0.5
Weight of XSs Associated with DS Boundary= 0.5
Percentile Method= 0
Sediment Output Level= 3
Mass or Volume Output= 0
Output Increment Type= 1
Profile and TS Output Increment= 1
XS Output Flag= 0
XS Output Increment= 10
Write Gradation File= 0
Read Gradation Hotstart= 0
Write HDF5 File= 1
Write Binary Output= 1
Write DSS Sediment File= 0
SV Curve= 0
Specific Gage Flag= 0

--- RENICKCK.f01 (steady flow) ---

Flow Title=Flow
Program Version=5.07
Number of Profiles= 6
Profile Names=f1p,f10p,f4p,f2p,f02p,f1pplus
River Rch & RM=ALUMRN,Main            ,13094
     682     363     481     579     950    1010
River Rch & RM=ALUMRN,Main            ,11059
     799     428     565     679    1110    1180
River Rch & RM=ALUMRN,Main            ,9883
     965     521     686     821    1340    1430
River Rch & RM=ALUMRN,Main            ,6456
    1080     584     767     917    1490    1590
River Rch & RM=ALUMRN,Main            ,284
    1350     740     968    1160    1860    2000
River Rch & RM=KTCHNCK,Main            ,41842
     743     397     525     631    1030    1100
River Rch & RM=KTCHNCK,Main            ,37328
     832     446     589     707    1150    1230
River Rch & RM=KTCHNCK,Main            ,35092
     926     499     657     788    1280    1370
River Rch & RM=KTCHNCK,Main            ,33009
    1030     557     732     876    1420    1520
River Rch & RM=KTCHNCK,Main            ,28691
    1150     622     817     977    1580    1700
River Rch & RM=KTCHNCK,Main            ,21556
    1810    1000    1300    1550    2480    2680
River Rch & RM=KTCHNCK,Main            ,16488
    2900    1630    2110    2490    3930    4290
River Rch & RM=KTCHNCK,Main            ,10721
    3870    2200    2830    3340    5220    5730
River Rch & RM=KTCHNCKT1,Main            ,9111
     634     336     447     537     884     938
River Rch & RM=KTCHNCKT1,Main            ,6856
     715     381     504     606     994    1060
River Rch & RM=KTCHNCKT1,Main            ,2501
     856     459     606     727    1190    1270
River Rch & RM=MILLCK1,Main            ,44569
     546     288     383     462     764     808
River Rch & RM=MILLCK1,Main            ,42192
     668     355     471     567     931     988
River Rch & RM=MILLCK1,Main            ,40676
     926     498     657     787    1280    1370
River Rch & RM=MILLCK1,Main            ,39243
    1580     868    1130    1350    2160    2330
River Rch & RM=MILLCK1,Main            ,32901
    1760     973    1270    1510    2410    2610
River Rch & RM=MILLCK1,Main            ,26603
    1970    1090    1420    1690    2700    2920
River Rch & RM=MILLCK1,Main            ,16549
    2620    1470    1890    2240    3550    3870
River Rch & RM=MILLCK1,Main            ,5376
    3090    1740    2250    2650    4180    4570
River Rch & RM=MILLCK1T1,Main            ,2820
     564     298     397     478     789     835
River Rch & RM=RENICKCK,Main            ,22028
     617     327     434     523     861     913
River Rch & RM=RENICKCK,Main            ,19013
     695     370     490     589     967    1030
River Rch & RM=RENICKCK,Main            ,16528
     937     505     665     797    1300    1390
River Rch & RM=RENICKCK,Main            ,13874
    1040     565     742     888    1440    1540
River Rch & RM=RENICKCK,Main            ,9049
    1170     638     837    1000    1620    1740
River Rch & RM=SNAKERN,Main            ,20697
     463     243     324     392     650     685
River Rch & RM=SNAKERN,Main            ,20190
     763     408     539     648    1060    1130
River Rch & RM=SNAKERN,Main            ,19342
     852     457     603     724    1180    1260
River Rch & RM=SNAKERN,Main            ,16967
    1190     644     845    1010    1630    1750
River Rch & RM=SNAKERN,Main            ,11910
    1330     728     952    1140    1830    1970
River Rch & RM=SNAKERN,Main            ,6596
    1480     812    1060    1260    2030    2190
Boundary for River Rch & Prof#=ALUMRN,Main            , 1
Up Type= 0
Dn Type= 3
Dn Slope=0.008838
Boundary for River Rch & Prof#=ALUMRN,Main            , 2
Up Type= 0
Dn Type= 3
Dn Slope=0.008838
Boundary for River Rch & Prof#=ALUMRN,Main            , 3
Up Type= 0
Dn Type= 3
Dn Slope=0.008838
Boundary for River Rch & Prof#=ALUMRN,Main            , 4
Up Type= 0
Dn Type= 3
Dn Slope=0.008838
Boundary for River Rch & Prof#=ALUMRN,Main            , 5
Up Type= 0
Dn Type= 3
Dn Slope=0.008838
Boundary for River Rch & Prof#=ALUMRN,Main            , 6
Up Type= 0
Dn Type= 3
Dn Slope=0.008838
Boundary for River Rch & Prof#=KTCHNCK,Main            , 1
Up Type= 0
Dn Type= 3
Dn Slope=0.005801
Boundary for River Rch & Prof#=KTCHNCK,Main            , 2
Up Type= 0
Dn Type= 3
Dn Slope=0.005801
Boundary for River Rch & Prof#=KTCHNCK,Main            , 3
Up Type= 0
Dn Type= 3
Dn Slope=0.005801
Boundary for River Rch & Prof#=KTCHNCK,Main            , 4
Up Type= 0
Dn Type= 3
Dn Slope=0.005801
Boundary for River Rch & Prof#=KTCHNCK,Main            , 5
Up Type= 0
Dn Type= 3
Dn Slope=0.005801
Boundary for River Rch & Prof#=KTCHNCK,Main            , 6
Up Type= 0
Dn Type= 3
Dn Slope=0.005801
Boundary for River Rch & Prof#=KTCHNCKT1,Main            , 1
Up Type= 0
Dn Type= 3
Dn Slope=0.024951
Boundary for River Rch & Prof#=KTCHNCKT1,Main            , 2
Up Type= 0
Dn Type= 3
Dn Slope=0.024951
Boundary for River Rch & Prof#=KTCHNCKT1,Main            , 3
Up Type= 0
Dn Type= 3
Dn Slope=0.024951
Boundary for River Rch & Prof#=KTCHNCKT1,Main            , 4
Up Type= 0
Dn Type= 3
Dn Slope=0.024951
Boundary for River Rch & Prof#=KTCHNCKT1,Main            , 5
Up Type= 0
Dn Type= 3
Dn Slope=0.024951
Boundary for River Rch & Prof#=KTCHNCKT1,Main            , 6
Up Type= 0
Dn Type= 3
Dn Slope=0.024951
Boundary for River Rch & Prof#=MILLCK1,Main            , 1
Up Type= 0
Dn Type= 3
Dn Slope=0.000839
Boundary for River Rch & Prof#=MILLCK1,Main            , 2
Up Type= 0
Dn Type= 3
Dn Slope=0.000839
Boundary for River Rch & Prof#=MILLCK1,Main            , 3
Up Type= 0
Dn Type= 3
Dn Slope=0.000839
Boundary for River Rch & Prof#=MILLCK1,Main            , 4
Up Type= 0
Dn Type= 3
Dn Slope=0.000839
Boundary for River Rch & Prof#=MILLCK1,Main            , 5
Up Type= 0
Dn Type= 3
Dn Slope=0.000839
Boundary for River Rch & Prof#=MILLCK1,Main            , 6
Up Type= 0
Dn Type= 3
Dn Slope=0.000839
Boundary for River Rch & Prof#=MILLCK1T1,Main            , 1
Up Type= 0
Dn Type= 3
Dn Slope=0.000001
Boundary for River Rch & Prof#=MILLCK1T1,Main            , 2
Up Type= 0
Dn Type= 3
Dn Slope=0.000001
Boundary for River Rch & Prof#=MILLCK1T1,Main            , 3
Up Type= 0
Dn Type= 3
Dn Slope=0.000001
Boundary for River Rch & Prof#=MILLCK1T1,Main            , 4
Up Type= 0
Dn Type= 3
Dn Slope=0.000001
Boundary for River Rch & Prof#=MILLCK1T1,Main            , 5
Up Type= 0
Dn Type= 3
Dn Slope=0.000001
Boundary for River Rch & Prof#=MILLCK1T1,Main            , 6
Up Type= 0
Dn Type= 3
Dn Slope=0.000001
Boundary for River Rch & Prof#=RENICKCK,Main            , 1
Up Type= 0
Dn Type= 3
Dn Slope=0.003087
Boundary for River Rch & Prof#=RENICKCK,Main            , 2
Up Type= 0
Dn Type= 3
Dn Slope=0.003087
Boundary for River Rch & Prof#=RENICKCK,Main            , 3
Up Type= 0
Dn Type= 3
Dn Slope=0.003087
Boundary for River Rch & Prof#=RENICKCK,Main            , 4
Up Type= 0
Dn Type= 3
Dn Slope=0.003087
Boundary for River Rch & Prof#=RENICKCK,Main            , 5
Up Type= 0
Dn Type= 3
Dn Slope=0.003087
Boundary for River Rch & Prof#=RENICKCK,Main            , 6
Up Type= 0
Dn Type= 3
Dn Slope=0.003087
Boundary for River Rch & Prof#=SNAKERN,Main            , 1
Up Type= 0
Dn Type= 3
Dn Slope=0.008894
Boundary for River Rch & Prof#=SNAKERN,Main            , 2
Up Type= 0
Dn Type= 3
Dn Slope=0.008894
Boundary for River Rch & Prof#=SNAKERN,Main            , 3
Up Type= 0
Dn Type= 3
Dn Slope=0.008894
Boundary for River Rch & Prof#=SNAKERN,Main            , 4
Up Type= 0
Dn Type= 3
Dn Slope=0.008894
Boundary for River Rch & Prof#=SNAKERN,Main            , 5
Up Type= 0
Dn Type= 3
Dn Slope=0.008894
Boundary for River Rch & Prof#=SNAKERN,Main            , 6
Up Type= 0
Dn Type= 3
Dn Slope=0.008894
DSS Import GetInterval= 0
DSS Import GetPeak= 0
DSS Import FillOption= 0

--- RENICKCK.g01 (geometry) ---

Geom Title=Geometry
Program Version=5.07

River Reach=RENICKCK        ,Main
Reach XY= 30
2074022.32474136316066.9551402932074278.95283702315519.694095716
2075019.65214303315039.0861330482075367.92310002314501.371985376
2076143.26013201314157.8392078732076795.34347352313431.797680959
2077200.55165261312885.4434587062077526.07265511311752.110095456
2077220.94170368310878.0760823792077409.35996202310666.850126877
2077145.83194578310478.5040468722077211.48929477309832.839327708
2076810.67283919309501.7389400452076578.06109968307878.341924384
2076189.09337369 307620.860155882076352.58386037306969.322088882
2075905.23928261306418.2559337912076185.44738361 305594.81860429
2076038.57234928305528.1517428762076079.71826437304405.235353544
2076276.07253045304273.464291632 2075976.5934706303854.193476632
2076163.57242736303435.9643262182075982.84345812  303355.7561533
2075964.09316751302520.8601852952076809.40578136301776.068367794
2076755.39112562301509.1578123722076902.00566179301707.074411288
2077165.80762762301609.6786087162077190.32496703301167.423915789

Type RM Length L Ch R = 1 ,22028   ,229.2,233.5,237.6
XS GIS Cut Line= 3
2074170.77752843 316082.63358663 2073993.6942212316049.647432134
2073686.40251294316035.758352295
#Sta/Elev= 30
       0  1868.5    42.2 1852.11    61.3 1845.33    89.5 1837.53   112.3 1832.33
   122.3 1829.18   125.6 1827.17   132.3 1820.74  134.281819.828   135.6 1819.22
   140.1 1818.55   152.3 1817.88   159.8 1818.72  163.75 1819.77     169 1821.97
   172.3 1822.42   180.1 1821.78   192.2 1821.59   218.4 1823.82   234.9  1822.6
   244.7 1821.19   280.8 1820.53   290.7 1821.07   307.1 1825.16   323.5 1826.29
   358.5 1827.75   405.7 1828.81   454.9 1830.77   474.4 1832.03   487.7 1830.76
#Mann= 3 ,-1 , 0
       0      .1       0  134.28    .045       0  163.75      .1       0
#XS Ineff= 2 , 0
                          171.48         1825.53
Permanent Ineff=
       F       F
Bank Sta=134.28,163.75
XS Rating Curve= 0 ,0
Exp/Cntr=0.3,0.1

Type RM Length L Ch R = 1 ,21794   ,311.1,312.7,311.6
XS GIS Cut Line= 3
2074223.15012711316005.3765233012074044.33093095315843.050076291
2073914.12252995315735.411183968
#Sta/Elev= 30
       0 1864.62    22.5 1856.18    42.3 1850.21    60.3 1846.55    76.2 1844.41
    91.1 1839.45    95.7 1837.17   117.9 1832.83   129.9  1827.4   137.5 1825.54
   154.3 1818.78   170.1 1816.51   178.7 1814.21   197.6 1815.54   210.9 1812.71
   215.4 1812.75   224.2  1815.6  254.031814.254   267.5 1812.25   272.4 1812.55
  275.281814.176   283.4 1822.37   293.3 1830.91   305.8 1838.39   316.6 1842.29
   367.9 1857.04   382.4 1862.17   391.6 1863.03   398.2  1865.8   410.4 1869.33
#Mann= 3 ,-1 , 0
       0      .1       0  254.03    .045       0  275.28      .1       0
Bank Sta=254.03,275.28
XS Rating Curve= 0 ,0
Exp/Cntr=0.3,0.1

Type RM Length L Ch R = 1 ,21482   ,278.1,278.4,277.7
XS GIS Cut Line= 3
2074432.35148036 315776.209986882074211.86537278 315595.65424563
2074144.15717486315538.362693548
#Sta/Elev= 30
       0 1873.91      10  1867.7    45.4 1849.19    55.8 1843.12    73.6  1830.3
    95.9 1810.81   102.9 1806.36   109.9 1804.87   116.9 1804.63   123.9 1805.09
     133 1807.64   149.5 1806.55   165.8 1807.64   183.9 1807.78   192.4 1804.44
   198.5 1805.41   205.9 1807.95   210.1 1808.04  216.191805.983   217.8 1805.11
   222.1 1804.63  232.571806.485   247.5 1806.71   268.7  1809.7     273 1812.03
   281.4 1819.51   305.7 1825.73   331.3 1837.77   354.7 1850.61   373.7 1856.91
#Mann= 3 ,-1 , 0
       0      .1       0  216.19    .045       0  232.57      .1       0
Bank Sta=216.19,232.57
XS Rating Curve= 0 ,0
Exp/Cntr=0.3,0.1

Type RM Length L Ch R = 1 ,21203   ,253.5,255.7,257.1
XS GIS Cut Line= 2
2074611.17100459315623.432077214 2074317.7683762315361.279386297
#Sta/Elev= 30
       0 1880.45     7.1  1875.5    25.7 1864.01    67.6 1841.11    94.5 1827.51
   119.2 1817.53   130.3 1812.25   144.2 1803.21     149  1801.2   153.5 1800.19
   179.8 1800.37   188.6 1799.78   202.9 1800.84   212.7 1800.27   222.6 1802.02
   227.5 1801.63   232.6 1800.49   247.2  1801.6   250.2 1801.11   254.6 1798.88
   263.4 1798.25   269.7 1798.94     279 1799.98   286.6 1801.82     303 1802.78
   320.6 1809.73   337.1 1814.15   365.4 1822.88   383.6 1829.65   393.5 1833.92
#Mann= 3 , 0 , 0
       0      .1       0   254.6    .045       0   269.7      .1       0
Bank Sta=254.6,269.7
XS Rating Curve= 0 ,0
Exp/Cntr=0.3,0.1

Type RM Length L Ch R = 1 ,20948   ,340.7,341.7,340.1
XS GIS Cut Line= 2
2074778.70577452315510.5848619642074486.17092651315132.980630293
#Sta/Elev= 30
       0 1912.07    24.1 1899.65    32.4 1893.88    41.5 1891.63    53.1 1884.43
    85.4 1866.81    94.6 1858.86   106.8 1849.95   152.7 1818.86   188.8 1798.24
   208.6 1794.46   219.1 1795.83   227.4 1794.69   240.3 1795.83   256.5 1793.69
   261.3 1795.18   273.1 1795.95   293.9 1795.41  302.111794.346  322.411795.017
   329.1 1796.84   347.9 1796.38   376.9 1797.12   401.8 1801.42   410.1 1803.69
   430.8 1813.69   455.4 1827.96   464.8 1835.05   471.1 1841.57   477.7 1846.52
#Mann= 3 ,-1 , 0
       0      .1       0  302.11    .045       0  322.41      .1       0
#XS Ineff= 2 , 0
                           332.2         1799.52
Permanent Ineff=
       F       F
Bank Sta=302.11,322.41
XS Rating Curve= 0 ,0
Exp/Cntr=0.3,0.1

Type RM Length L Ch R = 1 ,20606   ,306.6,303.3,297.8
XS GIS Cut Line= 2
 2074996.5875566315288.3625373842074737.03919119314922.911168545
#Sta/Elev= 30
       0 1903.88    28.5 1886.17    76.7 1854.21    92.6 1844.69   144.5 1811.71
   156.3 1805.09   170.4 1795.02  176.681789.378   177.6 1788.62   181.4 1787.71
   194.6 1787.23   200.3 1787.74  206.131789.365   209.5  1790.6   213.6 1791.09
   222.9 1790.26   229.7 1790.86   249.8 1790.47   257.8 1787.73   259.8 1787.73
   269.2 1789.97     290 1789.88   319.3 1788.86   334.3 1790.66   342.2 1792.65
   370.5 1802.37   410.7 1814.78   422.2 1816.85   431.6 1820.97   448.2 1825.98
#Mann= 3 ,-1 , 0
       0      .1       0  176.68    .045       0  206.13      .1       0
#XS Ineff= 2 , 0
                          287.21         1804.62
Permanent Ineff=
       F       F
Bank Sta=176.68,206.13
XS Rating Curve= 0 ,0
Exp/Cntr=0.3,0.1

Type RM Length L Ch R = 1 ,20303   ,365,369.9,372.2
XS GIS Cut Line= 3
2075254.40036118 315120.828095542075033.91425359314921.175279632
2074857.69872677314777.945907295
#Sta/Elev= 30
       0 1827.66    34.7 1826.42    67.2  1822.6    99.7 1813.61   132.5 1805.49
   136.9 1804.12   151.6 1796.95   166.2 1793.37     195 1791.06   256.4 1788.38
   297.2 1785.69   310.4 1783.62   318.2 1782.38   321.7 1782.78   323.6 1783.61
   329.8 1785.43   350.8 1785.76   365.9 1785.43   381.1 1784.15   393.5 1784.64
   406.8 1782.86   417.9 1784.17   423.1 1785.69   431.6 1786.54   441.8 1790.43
   456.9 1798.92   478.1 1809.67   507.1 1821.11   516.4 1823.32   524.5 1826.33
#Mann= 3 , 0 , 0
       0      .1       0   310.4    .045       0   323.6      .1       0
Bank Sta=310.4,323.6
XS Rating Curve= 0 ,0
Exp/Cntr=0.3,0.1

Type RM Length L Ch R = 1 ,19933   ,346.8,349.6,351
XS GIS Cut Line= 2
2075405.44172576314904.6822023842075175.40708086314539.230833545
#Sta/Elev= 30
       0 1839.87    23.7 1830.13    43.1 1819.89    50.9 1814.36    62.1 1811.62
    70.3 1806.52      78 1802.81   101.3 1794.77   124.5 1785.17   133.4 1780.35
   167.2 1780.92   184.6 1777.47   197.7 1778.89   209.2 1779.07   223.9 1777.81
   235.8 1778.23   248.6 1777.66   260.2 1775.92   271.9 1776.45   285.7 1775.26
  296.82 1775.49   309.5 1774.56   313.9 1775.09  316.841776.428   321.4 1779.04
   326.1 1782.81   332.4 1785.18   380.9 1795.07   402.3 1803.49   431.8 1818.69
#Mann= 3 ,-1 , 0
       0      .1       0  296.82    .045       0  316.84      .1       0
#XS Ineff= 2 , 0
           269.1 1781.87
Permanent Ineff=
       F       F
Bank Sta=296.82,316.84
XS Rating Curve= 0 ,0
Exp/Cntr=0.3,0.1

Type RM Length L Ch R = 1 ,19583   ,272.9,274.2,273.7
XS GIS Cut Line= 2
2075636.97768003 314709.442107292075454.68604985314331.837875634
#Sta/Elev= 30
       0 1822.75    53.2 1805.35    71.5 1801.16      86 1797.09   115.2 1790.63
   122.5 1788.38   135.5 1786.72   144.3 1783.38   157.6 1781.91   162.5 1780.97
   169.8 1777.55   173.5 1776.59   187.1 1776.37   220.8 1773.07   246.1 1772.11
   253.1 1771.27   260.8 1769.72  268.621769.793   275.5  1768.9     290 1768.24
  301.37 1769.57   304.6 1770.66   313.5 1772.38   324.5 1777.62   344.7  1785.3
     352  1788.5   373.8 1799.81     396 1809.45   410.7 1817.65   419.3 1823.84
#Mann= 3 ,-1 , 0
       0      .1       0  268.62    .045       0  301.37      .1       0
Bank Sta=268.62,301.37
XS Rating Curve= 0 ,0
Exp/Cntr=0.3,0.1

Type RM Length L Ch R = 1 ,19309   ,300.5,296.2,290.5
XS GIS Cut Line= 2
2075872.43783903314603.105049625 2075678.2102091314174.502560377
#Sta/Elev= 30
       0 1857.83      31  1842.2    76.4 1822.25    97.8 1814.43   126.8  1805.5
   192.1 1783.23   202.4  1777.5     207 1776.54   221.9 1775.65   224.4 1774.93
   234.3 1769.56   239.2 1768.03   252.9 1766.86   263.7  1767.1   267.3 1766.29
  269.611764.955   274.5 1763.27   281.7 1763.07   288.9 1763.28   296.1 1764.97
   296.2 1765.02   301.2 1766.21   338.4 1767.59   360.9 1773.04     384 1784.77
   422.6 1807.34     435  1813.3   443.8 1815.38     451 1820.08   470.6 1828.68
#Mann= 4 ,-1 , 0
       0      .1       0  269.61    .045       0   296.1    .045       0
   296.2      .1       0
#XS Ineff= 2 , 0
          262.94 1768.14
Permanent Ineff=
       F       F
Bank Sta=269.61,296.1
XS Rating Curve= 0 ,0
Exp/Cntr=0.3,0.1

Type RM Length L Ch R = 1 ,19013   ,281.3,278,270.3
XS GIS Cut Line= 3
2076207.72424194314425.153633878 2075984.1997546314195.118988961
2075835.54519626314041.039244622
#Sta/Elev= 30
       0 1852.56    36.4 1841.92    77.6 1826.82   151.9 1792.89   179.7 1779.33
   200.6 1770.21   212.2 1765.96   218.9  1762.6   223.8 1761.69   235.4 1761.12
  248.741758.368   270.7 1757.24   278.21758.368   281.8 1760.18   291.1 1767.76
   297.2 1771.22   320.1 1776.85   341.4  1779.8   365.3 1780.03   376.9 1782.57
   407.6 1782.97   426.5 1783.92   431.2  1784.9   445.4 1789.33   454.8  1795.8
   469.8 1801.84   476.7  1805.4   484.2 1807.65   523.1 1827.73   534.8 1832.78
#Mann= 3 ,-1 , 0
       0      .1       0  248.74    .045       0   278.2      .1       0
Bank Sta=248.74,278.2
XS Rating Curve= 0 ,0
Exp/Cntr=0.3,0.1

Type RM Length L Ch R = 1 ,18735   ,248.2,248.9,250.1
XS GIS Cut Line= 2
2076451.86482978314158.2266742892076046.04871228313960.744129628
#Sta/Elev= 30
       0 1854.76    13.6 1849.88    25.2 1843.64    36.2 1841.23    47.1 1835.53
    55.3 1832.87   153.4 1791.84   182.9 1781.24   192.7 1775.31   209.9 1774.09
   218.6 1769.12   229.7 1764.72   240.5 1757.27   251.6 1751.76  261.091750.143
   280.6 1748.21   288.4 1748.91   293.3 1750.52   300.7 1754.22     313 1755.54
   320.8 1758.75   335.4 1768.24   369.4 1793.43   401.1 1813.39   415.6 1824.78
   422.9 1827.56   433.2 1829.43   438.2 1831.82   444.8 1836.48   451.3 1837.92
#Mann= 3 , 0 , 0
       0      .1       0  261.09    .045       0   293.3      .1       0
Bank Sta=261.09,293.3
XS Rating Curve= 0 ,0
Exp/Cntr=0.3,0.1

Type RM Length L Ch R = 1 ,18486   ,249.5,252.3,256.3
XS GIS Cut Line= 2
2076557.11658779313950.9784011242076204.46899912313753.495856464
#Sta/Elev= 30
       0 1799.85    22.6 1793.36    33.8  1787.5    41.4 1785.24    63.4 1781.84
      94 1780.65    97.5 1779.38   103.6  1775.9   119.2 1771.31   127.8 1767.05
   142.9  1766.2   160.1 1758.32   176.7  1752.4   184.2 1750.37   197.6 1748.18
   233.1 1745.64  239.641744.107   248.2 1743.17   259.4 1743.28  267.281744.172
   274.5 1747.15   295.1 1747.37   297.5 1748.07   302.3 1750.91   319.6 1765.61
   334.7 1781.14   349.7 1793.13     376 1816.56   389.1 1825.55   404.2 1834.68
#Mann= 3 ,-1 , 0
       0      .1       0  239.64    .045       0  267.28      .1       0
#XS Ineff= 2 , 0
                          275.89         1749.92
Permanent Ineff=
       F       F
Bank Sta=239.64,267.28
XS Rating Curve= 0 ,0
Exp/Cntr=0.3,0.1

Type RM Length L Ch R = 1 ,18234   ,325,327.8,329.3
XS GIS Cut Line= 2
2076699.26066044313824.0252429542076399.78127253313539.737097621
#Sta/Elev= 30
       0 1790.83    17.8 1782.82    42.2 1773.57    60.3 1770.26    82.9 1763.66
   106.9 1752.12   119.1 1751.66     137 1747.52   153.3 1745.46   165.5 1745.22
   178.8 1742.51     205  1741.3   218.6 1742.43   223.1 1742.06   232.2 1738.97
   250.3 1740.42  255.621738.946   260.1 1737.42     267 1736.95  278.791738.483
   283.3 1741.33   289.4 1748.96   297.2 1756.66   322.6 1773.34     339 1780.38
   346.6 1785.27   372.4 1797.95   381.4 1800.68   399.5 1812.31   412.9 1819.07
#Mann= 3 ,-1 , 0
       0      .1       0  255.62    .045       0  278.79      .1       0
Bank Sta=255.62,278.79
XS Rating Curve= 0 ,0
Exp/Cntr=0.3,0.1

Type RM Length L Ch R = 1 ,17906   ,380.5,382.2,376.3
XS GIS Cut Line= 2
2076943.40124828313695.987113208 2076676.4742887313324.893367216
#Sta/Elev= 30
       0 1795.48    43.3 1777.02    75.6 1764.17    83.7 1757.86      88 1756.72
    99.9    1756     108  1750.1   116.2 1749.24   120.1 1748.04   132.7 1740.89
   144.4 1740.68   156.2  1736.9   172.6  1735.5   200.9 1734.97   250.2 1735.59
   262.6 1734.33   285.8 1735.25  293.861734.817   297.9 1733.39   301.9 1733.09
  316.721733.909   330.1 1734.78   352.5 1733.97   358.4 1736.12   381.9 1754.79
   390.9 1762.82   398.3 1767.22     407 1775.05   447.4 1805.64   457.1 1812.05
#Mann= 3 ,-1 , 0
       0      .1       0  293.86    .045       0  316.72      .1       0
#XS Ineff= 2 , 0
          209.68 1743.49
Permanent Ineff=
       F       F
Bank Sta=293.86,316.72
XS Rating Curve= 0 ,0
Exp/Cntr=0.3,0.1

Type RM Length L Ch R = 1 ,17524   ,281.5,277.3,273
XS GIS Cut Line= 2
2077339.45163727313476.8031683712076878.29704776313065.561864883
#Sta/Elev= 30
       0 1819.82    28.4 1811.37    58.7 1798.37    89.9 1780.99   133.3 1752.88
   160.2 1740.78     169 1738.34     177 1737.29   216.4 1737.31   248.2  1736.5
   265.7    1735   278.9 1735.47   309.7 1733.06   336.1  1733.7   364.3 1732.17
   384.4 1730.07     454 1728.75   467.51726.595   474.9 1724.71   487.6 1724.04
   492.5 1724.35  495.681726.759   503.1 1736.56   507.5 1741.34   517.1 1749.31
   531.9 1763.72   538.3 1768.61   564.7 1776.77     598 1785.29   617.9 1792.04
#Mann= 3 ,-1 , 0
       0      .1       0   467.5    .045       0  495.68      .1       0
Bank Sta=467.5,495.68
XS Rating Curve= 0 ,0
Exp/Cntr=0.3,0.1

Type RM Length L Ch R = 1 ,17246   ,355.6,353.8,351.6
XS GIS Cut Line= 2
2077466.40479544313092.6884510522077052.99322069312902.801363632
#Sta/Elev= 30
       0 1793.36      33 1780.34    58.3 1772.29    72.7 1767.12      80 1765.51
   103.9 1755.03   126.1 1742.82   141.3 1735.19     163 1729.32   166.6 1728.95
   173.8 1729.38   195.4 1727.71   202.7 1727.76   220.8 1724.92   237.4 1723.55
   252.3 1724.49   267.1 1724.68   274.6 1724.15     311 1723.84   314.1 1722.68
   318.3 1721.76   332.7 1721.48   338.9 1721.82   342.7 1722.64   350.7 1725.64
     356 1729.45   366.1 1735.46   404.9 1756.01   435.4    1776   454.9 1790.87
#Mann= 3 , 0 , 0
       0      .1       0   314.1    .045       0   342.7      .1       0
Bank Sta=314.1,342.7
XS Rating Curve= 0 ,0
Exp/Cntr=0.3,0.1

Type RM Length L Ch R = 1 ,16892   ,365.8,364.8,363.1
XS GIS Cut Line= 2
2077608.54886812312718.3394622062077125.69287845312577.280361131
#Sta/Elev= 30
       0 1786.15    11.9 1779.54    22.1 1777.21    39.2 1768.55    46.1 1766.28
      72 1754.22    90.5 1742.39     111 1726.99   122.2 1721.05   128.1  1719.2
   148.6  1717.1   172.5 1719.06   199.9 1718.82   209.5 1718.07   219.1 1719.41
   238.6 1717.74   288.7 1720.15  336.26 1718.88  356.311719.276   360.5 1720.53
   377.6 1735.76   394.7 1760.87   398.1 1764.43   404.9 1769.59   411.8 1773.85
   439.1 1788.39   463.4 1800.06   473.3  1805.8   487.2 1811.86     503 1817.63
#Mann= 3 ,-1 , 0
       0      .1       0  336.26    .045       0  356.31      .1       0
Bank Sta=336.26,356.31
XS Rating Curve= 0 ,0
Exp/Cntr=0.3,0.1

Type RM Length L Ch R = 1 ,16528   ,330.1,327.8,324.8
XS GIS Cut Line= 2
2077725.30224353312328.4741002172077176.69113603312248.613039464
#Sta/Elev= 30
       0 1781.71    20.1 1771.28    43.3 1761.94    89.7 1747.81     103 1742.38
   112.9 1740.25   126.2 1733.93   146.1 1721.91   159.3 1715.55   182.6 1713.63
   205.8 1713.81   222.3  1711.6   238.9 1712.06   245.5 1713.45   262.1 1713.22
   275.4 1710.97   288.6 1713.91   315.2 1715.72   325.1 1715.29   330.5 1713.02
   344.3  1713.2   351.6 1714.06   364.9 1713.34   368.2 1714.63   378.2 1723.45
   419.5 1769.89   431.2 1780.85   493.4 1823.49   536.1 1847.26   554.4 1855.16
#Mann= 3 , 0 , 0
       0      .1       0   330.5    .045       0   344.3      .1       0
Bank Sta=330.5,344.3
XS Rating Curve= 0 ,0
Exp/Cntr=0.3,0.1

Type RM Length L Ch R = 1 ,16200   ,331.8,328.9,319.6
XS GIS Cut Line= 2
2077728.77434945311983.8560230432077279.12170544311967.362945795
#Sta/Elev= 30
       0 1765.96    23.4 1750.26    43.1  1739.7    62.8 1730.39    82.5 1724.11
   115.3 1716.97   125.1 1713.97   161.3 1713.17   200.7 1710.15   236.8 1709.81
   243.3 1709.13   253.2 1709.88  259.03 1707.48     263 1706.15   276.2 1705.87
   282.7 1706.18     286 1707.23   289.3    1709   292.6 1709.79   302.4  1709.3
   322.1 1710.45   332.4  1714.2     355 1720.53   384.5 1731.32   400.9 1738.87
   410.8 1742.34   423.9 1749.59   433.8 1753.03   440.3 1757.24     450  1762.5
#Mann= 3 , 0 , 0
       0      .1       0  259.03    .045       0     286      .1       0
Bank Sta=259.03,286
XS Rating Curve= 0 ,0
Exp/Cntr=0.3,0.1

Type RM Length L Ch R = 1 ,15871   ,263.4,266.3,269.2
XS GIS Cut Line= 2
2077675.82301179311594.0989285412077182.76756743 311801.56439288
#Sta/Elev= 30
       0 1765.63    56.9  1750.4    92.5 1742.82   113.8 1739.68   128.1 1736.58
   155.1 1726.13   167.7 1719.97   170.8 1717.76   174.3 1712.99   177.9 1706.87
   181.5 1703.84   192.7 1702.51   202.8 1702.92   206.4 1703.93   209.9 1705.35
   213.5 1705.63   227.8 1703.88   234.9 1704.41     242 1706.17   277.6 1707.57
   330.5 1706.16     348 1707.02   360.6 1704.66   370.1 1706.78   405.7 1706.53
   420.7 1707.45   427.1 1710.34   434.2 1715.67   490.8 1766.11   534.9 1801.96
#Mann= 3 , 0 , 0
       0      .1       0   181.5    .045       0   206.4      .1       0
Bank Sta=181.5,206.4
XS Rating Curve= 0 ,0
Exp/Cntr=0.3,0.1

Type RM Length L Ch R = 1 ,15605   ,379.4,378.9,374.8
XS GIS Cut Line= 2
2077676.69112027311389.2377897052077061.23992336311461.286530122
#Sta/Elev= 30
       0 1789.58    70.2 1749.79    83.4 1743.07    99.9 1736.42   119.7 1731.62
   162.7  1725.3   179.2 1720.01   195.7 1710.43   212.2    1704  264.921701.096
     275 1699.28  285.011701.145   294.8 1701.85   321.2 1700.59   327.8  1702.4
     341 1702.74   397.2 1701.57     417 1702.99   440.1 1702.98   448.4 1704.89
   473.2 1717.36     493  1729.5   502.9 1737.01   519.3 1751.88   542.5 1771.27
   551.9 1777.31   575.5 1796.19   585.5 1801.63   599.2  1813.5   619.7  1828.6
#Mann= 3 ,-1 , 0
       0      .1       0  264.92    .045       0  285.01      .1       0
Bank Sta=264.92,285.01
XS Rating Curve= 0 ,0
Exp/Cntr=0.3,0.1

Type RM Length L Ch R = 1 ,15226   ,627.7,631.8,628.1
XS GIS Cut Line= 3
2077661.06615153310983.8560545442077280.85792243311121.876775876
2077088.14964643311184.376978964
#Sta/Elev= 30
       0  1770.9    26.1 1762.34    43.6 1754.37    57.5 1746.57    64.5 1740.51
    78.5 1737.67    88.9 1729.64   113.4 1715.42   120.4 1712.72   162.2 1708.95
   183.2 1698.53   266.9 1698.44  271.691697.064   284.4 1695.67  291.741696.708
   308.4  1698.3   326.3 1697.63   346.8 1698.64   354.2 1700.39   364.8 1705.59
   375.1 1708.67   434.1  1718.9   465.2 1717.99     479  1714.7   489.1 1718.86
   503.1 1727.55   516.9 1733.93     541 1742.88   592.8 1758.29   607.1 1764.75
#Mann= 3 ,-1 , 0
       0      .1       0  271.69    .045       0  291.74      .1       0
Bank Sta=271.69,291.74
XS Rating Curve= 0 ,0
Exp/Cntr=0.3,0.1

Type RM Length L Ch R = 1 ,14594   ,339.4,342.4,343.6
XS GIS Cut Line= 3
2077598.34908536310600.1753914652077366.14416918310676.130292043
2077005.90112329310821.529607549
#Sta/Elev= 30
       0 1751.59      20 1748.32    50.1 1738.66    70.9 1730.53    94.3 1724.12
   108.3  1718.4     129 1707.75   153.1  1701.8   173.9 1699.04   184.2 1696.59
   190.4 1692.02     198 1690.34  210.511691.751   229.1  1691.6   239.4 1693.09
   267.6 1693.65   356.1 1693.85   444.5 1693.66   454.4 1694.74   458.7 1696.25
   465.8 1699.87   483.4 1713.87   490.5 1718.66   514.9 1729.48   525.9 1736.01
   540.1 1746.12   557.7 1760.69   575.3 1773.52     625 1807.71   632.8 1811.83
#Mann= 5 ,-1 , 0
       0      .1       0   173.9     .05       0   190.4    .045       0
  210.51     .05       0   356.1      .1       0
Bank Sta=190.4,210.51
XS Rating Curve= 0 ,0
Exp/Cntr=0.3,0.1

Type RM Length L Ch R = 1 ,14251   ,380.4,377.9,370.6
XS GIS Cut Line= 2
2077560.37179911310426.5641901342076966.83886543310494.923633456
#Sta/Elev= 30
       0 1770.93     9.2 1767.17    42.2  1751.4    68.7 1741.74    81.9 1737.73
    91.8 1732.04   101.7 1731.45   118.2 1723.39   141.3 1708.98   164.4 1700.04
   173.5 1695.17   180.9 1692.72     218 1689.16   240.4  1690.3   256.9 1689.77
   286.6 1690.79   346.1 1689.99     356  1690.7  407.861690.214   418.7 1688.59
  427.881689.647   438.5 1690.81     449 1690.96   463.8 1688.78   484.8 1691.94
   488.1 1693.86     498 1701.62   511.1 1710.25   540.8  1728.4   597.5  1772.8
#Mann= 6 ,-1 , 0
       0      .1       0    7.03      .1       0  246.32     .05       0
  367.77      .1       0  407.86    .045       0  427.88      .1       0
Bank Sta=407.86,427.88
XS Rating Curve= 0 ,0
Exp/Cntr=0.3,0.1

Type RM Length L Ch R = 1 ,13874   ,377.9,377.2,370.6
XS GIS Cut Line= 2
2077434.50361252 310114.064487042076984.19972309310278.994931459
#Sta/Elev= 30
       0 1744.82    31.9 1734.64    39.6 1733.48    53.9 1729.19    78.4 1719.88
    92.3 1718.76    98.4 1716.37   106.3 1714.38   131.7 1705.25   144.7 1698.16
   151.7 1692.94   155.2 1691.05  169.641685.638   172.7 1684.59   183.2 1683.03
  195.741685.124   211.1 1687.38     220    1688   235.6 1687.26     260 1687.77
   270.5 1687.24   284.5 1688.48   315.8    1689   350.9 1692.66   392.5  1695.8
   410.8  1700.2   441.7 1710.63   452.2 1712.29   466.2 1716.66   479.6  1719.1
#Mann= 6 ,-1 , 0
       0      .1       0      25      .1       0  169.64    .045       0
  195.74      .1       0  246.94     .05       0  325.03      .1       0
Bank Sta=169.64,195.74
XS Rating Curve= 0 ,0
Exp/Cntr=0.3,0.1

Type RM Length L Ch R = 1 ,13496   ,404.3,408,406.9
XS GIS Cut Line= 2
2077347.69801185309704.9931267052076843.14095011310077.171844289
#Sta/Elev= 30
       0 1800.15    26.2 1782.26    36.6 1774.22    52.9 1764.27    60.3 1758.28
    69.7 1753.05    98.1 1734.07   101.8 1732.38   109.6 1731.87   114.3 1730.43
   125.7 1723.46   133.1 1720.99   142.6 1715.61   163.6 1699.06  177.581683.487
     180 1682.15   186.5  1681.2  202.461683.583   232.2 1682.49   309.7 1684.55
     326 1683.06   339.5 1684.39   403.5 1683.31   489.7 1684.17   505.4 1687.77
   529.2 1696.45   567.1 1705.36     591 1714.42     607 1719.18     627 1727.74
#Mann= 6 ,-1 , 0
       0      .1       0  154.29      .1       0  177.58    .045       0
  202.46      .1       0  374.92     .05       0  448.69      .1       0
Bank Sta=177.58,202.46
XS Rating Curve= 0 ,0
Exp/Cntr=0.3,0.1

Type RM Length L Ch R = 1 ,13088   ,367.1,374.2,373.9
XS GIS Cut Line= 2
2077030.85776627309484.7242102922076595.74511945 309778.77775605
#Sta/Elev= 30
       0 1719.97     5.5 1719.07    19.6 1714.07    34.5 1714.27    45.5 1709.79
    88.7 1697.33   100.6 1693.36   108.5 1688.81   116.4 1682.99   120.4  1681.5
  176.141678.532   183.7  1677.1   199.6 1676.81   203.5 1677.05   205.51678.034
   207.5  1679.2   213.3 1680.12   239.1 1679.75     251 1680.53   340.9 1680.08
     350 1678.18   364.5    1681   374.3 1686.97   397.6 1695.82   414.2 1705.84
   421.3 1710.99   432.9 1720.68   459.1 1738.85   480.3 1757.31   525.2 1794.09
#Mann= 7 ,-1 , 0
       0      .1       0  141.18     .05       0  156.67      .1       0
  176.14    .045       0   205.5      .1       0  266.12     .05       0
  376.99      .1       0
Bank Sta=176.14,205.5
XS Rating Curve= 0 ,0
Exp/Cntr=0.3,0.1

Type RM Length L Ch R = 1 ,12714   ,385.3,386.6,385.1
XS GIS Cut Line= 2
2076985.28502277309226.4776795512076516.53497604309384.897638291
#Sta/Elev= 30
       0 1742.41     5.2 1738.57    12.1 1731.03    15.6 1728.49    26.1  1725.5
    32.9 1722.07    44.3 1712.75    64.1 1694.38    81.4 1681.44    85.7 1678.83
    91.8 1677.24   105.6 1676.75   158.1  1678.3     168 1677.92   178.4 1675.64
  186.781675.306   202.6 1673.85  219.551675.785   226.8 1675.57   230.3 1676.67
   237.2  1677.2   264.9 1677.56   303.1 1679.22   320.4 1680.39   344.3  1683.8
   354.9 1685.74   368.8 1689.51   393.1 1698.08   438.1 1705.71   494.8 1716.79
#Mann= 6 ,-1 , 0
       0      .1       0   39.77      .1       0  140.47     .05       0
  186.78    .045       0  219.55     .05       0  297.31      .1       0
Bank Sta=186.78,219.55
XS Rating Curve= 0 ,0
Exp/Cntr=0.3,0.1

Type RM Length L Ch R = 1 ,12328   ,394.1,401.3,402.3
XS GIS Cut Line= 2
2076839.88570726308896.6164626332076339.66853186  309063.7171783
#Sta/Elev= 30
       0 1735.43       6 1730.22    14.5 1724.14    28.3 1716.69    49.1 1703.61
    52.5 1702.83    59.4 1702.33    62.9 1701.44    66.4 1699.74    76.7 1692.34
      94 1683.49    97.5 1682.59   107.9 1681.61   121.7 1676.97   135.5 1674.22
   142.5  1673.6  160.511673.242   173.6 1671.79   187.8 1672.53  193.271673.519
   201.3 1674.33   242.8  1673.7   345.7 1673.61   388.1 1674.86   415.7 1676.69
   439.9 1681.76   464.2 1689.44   481.5 1695.98   514.5 1709.87   527.4 1716.98
#Mann= 7 ,-1 , 0
       0      .1       0   79.47      .1       0  121.56      .1       0
  160.51    .045       0  193.27      .1       0  301.47     .05       0
  453.22      .1       0
Bank Sta=160.51,193.27
XS Rating Curve= 0 ,0
Exp/Cntr=0.3,0.1

Type RM Length L Ch R = 1 ,11926   ,549.8,556,548.1
XS GIS Cut Line= 2
2076816.01403585308617.7535032932076221.39613062308575.436002627
#Sta/Elev= 30
       0 1741.44    12.9 1734.88    19.4 1732.43    45.8 1725.43    52.3  1721.2
    65.5 1718.74    75.4 1713.35   121.4 1694.15   134.6 1689.35   144.4 1684.04
   154.3 1677.28   170.7 1669.71   190.5 1670.56   222.11669.128   233.2 1667.57
   236.5 1667.78  242.161669.778   249.7  1670.7   285.9 1671.42   305.6 1669.52
   318.7 1670.25   351.6 1669.39   394.4 1669.98   430.6 1673.03   446.3 1677.07
   476.6 1682.66   483.2 1685.44   532.5  1698.3     552 1704.74   596.1 1717.56
#Mann= 8 ,-1 , 0
       0      .1       0   70.87      .1       0  196.33     .05       0
   222.1    .045       0  242.16     .05       0   391.5      .1       0
  524.39     .05       0  532.48      .1       0
Bank Sta=222.1,242.16
XS Rating Curve= 0 ,0
Exp/Cntr=0.3,0.1

Type RM Length L Ch R = 1 ,11370   ,461.4,451.1,434.9
XS GIS Cut Line= 2
2076780.20669279308124.0471416262076150.86641604308142.493298963
#Sta/Elev= 30
       0  1765.6    36.1 1744.34    52.5 1731.86    78.8 1713.73    95.2 1697.99
     105 1691.67   118.1 1685.24   141.1 1676.31   154.3 1669.99   173.9 1669.08
   183.7 1667.07   193.6 1666.13  226.341665.118   229.7 1663.99   236.3 1663.28
   242.9 1663.49   246.2 1664.22  247.861665.429   252.7 1668.54     256 1669.31
     279 1671.05   354.5 1673.11   403.7 1675.93   433.2 1678.87   469.3 1679.17
   515.3 1681.53   535.5 1688.18   563.2 1695.59   589.6 1703.77   629.6 1712.78
#Mann= 6 ,-1 , 0
       0      .1       0   13.49      .1       0  118.88      .1       0
  199.65     .05       0  226.34    .045       0  247.86     .05       0
Bank Sta=226.34,247.86
XS Rating Curve= 0 ,0
Exp/Cntr=0.3,0.1

Type RM Length L Ch R = 1 ,10919   ,362.7,378.3,383.5
XS GIS Cut Line= 2
2076569.70317677307602.1285660422076115.05907294308116.451356292
#Sta/Elev= 30
       0 1727.45     4.1 1724.17      19 1717.32    45.4 1702.67    61.7 1696.62
    68.6 1692.25    73.1 1690.52    83.4 1689.88    94.2 1685.86   110.5 1680.96
     123 1675.68   145.3 1672.71   167.6 1665.11  196.13 1663.01   204.5 1660.76
   210.4 1660.55  232.091662.532   270.2 1663.09   296.4 1665.72   504.5 1670.39
     546 1672.34   563.6 1675.68   570.7 1677.68   584.6 1683.81   596.3 1684.11
   600.9  1684.9   610.2 1689.28   656.7  1706.4     673 1711.58   686.5 1714.83
#Mann= 4 ,-1 , 0
       0      .1       0  155.92     .05       0  196.13    .045       0
  232.09     .05       0
Bank Sta=196.13,232.09
XS Rating Curve= 0 ,0
Exp/Cntr=0.3,0.1

Type RM Length L Ch R = 1 ,10541   ,358.5,361.6,358.8
XS GIS Cut Line= 2
2076563.19301918307535.9393939672075802.55936986307532.684151128
#Sta/Elev= 30
       0 1733.68    12.6 1724.48    45.2 1703.52    61.8 1694.69    97.9 1682.69
   114.3 1681.23   137.5  1676.9   143.9 1674.36   160.5 1665.15   166.5 1663.25
   195.9 1661.32   222.6 1662.04   271.8 1660.34   288.2 1661.41   327.6 1661.72
   334.2 1661.51  335.671660.575   340.7 1658.51     344 1658.33  360.141660.316
   435.9 1664.26   494.9  1668.7   540.8 1672.89   573.7    1677   599.9 1681.23
     659 1693.07   675.4 1699.47   698.3 1698.99   734.4 1712.24   760.6 1724.49
#Mann= 5 ,-1 , 0
       0      .1       0  159.35     .05       0  335.67    .045       0
  360.14     .05       0  562.96      .1       0
Bank Sta=335.67,360.14
XS Rating Curve= 0 ,0
Exp/Cntr=0.3,0.1

Type RM Length L Ch R = 1 ,10179   ,408.9,411.9,409.6
XS GIS Cut Line= 2
2076480.72763294307275.5225919632075879.59924203307254.906491458
#Sta/Elev= 30
       0 1720.08     8.9 1713.11      22 1700.59    41.7 1689.76    48.3 1685.52
    58.2 1683.96    81.1 1675.11    93.5 1671.38   110.7 1668.85   127.1 1665.41
   136.9 1661.28   143.5  1659.2   156.6 1658.25   238.7 1659.18     265 1658.69
   278.1 1659.25  292.111658.582   301.1 1656.73   310.9 1656.78  315.361658.468
   320.8 1659.73   402.8 1660.97   412.7 1661.87   422.5 1664.29   488.2 1684.38
     521  1692.4   560.4 1700.88   583.4 1700.19   593.2 1704.66   601.5 1706.88
#Mann= 5 ,-1 , 0
       0      .1       0  104.34     .05       0  292.11    .045       0
  315.36     .05       0  502.62      .1       0
Bank Sta=292.11,315.36
XS Rating Curve= 0 ,0
Exp/Cntr=0.3,0.1

Type RM Length L Ch R = 1 ,9767    ,709.9,718.4,695.7
XS GIS Cut Line= 3
2076500.54813135306989.7154207972076302.63153243306986.243314877
2075868.60385719306977.562557966
#Sta/Elev= 30
       0 1724.31    22.2 1715.42    49.6 1700.22    80.6 1686.83   107.5 1669.53
   120.6 1664.16   127.2 1662.26   130.5 1660.37   133.7 1657.19  135.681655.989
     137  1655.2   143.6 1654.45  155.691655.875   175.4 1656.93     219 1656.28
   232.2 1655.15   245.3 1656.23   258.4 1656.38   324.1 1655.02   343.7  1656.6
   360.2 1657.03   502.2 1656.06   547.2 1657.99   563.6 1659.09   579.2 1661.98
   593.7 1667.51   606.3 1675.69   612.8  1680.8   616.1 1682.29   632.1 1681.82
#Mann= 6 ,-1 , 0
       0      .1       0   18.64      .1       0  135.68    .045       0
  155.69      .1       0  169.71     .05       0   573.3      .1       0
Bank Sta=135.68,155.69
XS Rating Curve= 0 ,0
Exp/Cntr=0.3,0.1

Type RM Length L Ch R = 1 ,9049    ,613.6,618.3,611.8
XS GIS Cut Line= 2
 2076477.9786227306564.3681743742075858.18721136 306618.18762055
#Sta/Elev= 30
       0 1691.33    42.8 1682.54    75.3 1676.51    85.2 1673.79   114.8 1669.41
   144.5 1663.51   157.2 1661.81   213.6 1659.47   299.3 1654.84     319 1654.78
   328.9  1653.8   369.3 1653.96  388.821652.761   398.1 1650.92   404.7 1650.53
   414.8 1651.18  422.391652.606   429.9 1653.68   440.9 1653.84   463.2 1653.27
   480.4 1653.52   490.3 1652.44   503.4 1653.61   549.6    1653   556.1 1655.02
   566.3 1659.98   592.4 1673.67   602.6  1680.7   605.5 1681.82   622.1 1681.52
#Mann= 5 ,-1 , 0
       0      .1       0  119.24     .05       0  388.82    .045       0
  422.39     .05       0  511.12      .1       0
Bank Sta=388.82,422.39
XS Rating Curve= 0 ,0
Exp/Cntr=0.3,0.1

Type RM Length L Ch R = 1 ,8431    ,613.8,626.2,620.7
XS GIS Cut Line= 2
2076408.53420776306086.9376987962075806.10365412306128.604282126
#Sta/Elev= 30
       0 1708.11    15.5  1697.3    28.6    1692    58.2  1677.8    68.1 1675.09
    83.8 1667.53   104.3 1660.36   130.6 1654.04   173.3 1649.78   189.8 1650.56
     295 1649.98   304.9 1650.72   347.6 1650.87  352.531649.964   357.5 1648.53
   360.8 1648.34  381.911649.982   396.3  1650.9   436.4 1651.07   449.8 1649.84
   505.5 1651.38   512.1 1652.91   521.9 1656.47   538.4 1664.46   544.7 1666.78
     568 1673.03   585.2 1679.55   594.3  1684.1   597.6 1685.13   603.9 1685.69
#Mann= 5 ,-1 , 0
       0      .1       0  177.23     .05       0  352.53    .045       0
  381.91     .05       0  509.62      .1       0
Bank Sta=352.53,381.91
XS Rating Curve= 0 ,0
Exp/Cntr=0.3,0.1

Type RM Length L Ch R = 1 ,7805    ,528.9,544.1,535
XS GIS Cut Line= 2
2076405.06210187305741.4515131262075793.95111936305665.062558293
#Sta/Elev= 30
       0  1719.4     8.8 1710.01      22 1699.32    38.5 1691.17    61.7 1683.17
    68.3 1679.47    91.4 1663.69   101.3 1657.88   104.7  1656.7   134.4  1651.6
   193.9  1647.2   203.8 1648.17     260 1648.38  294.831646.632     303 1644.27
     313  1645.1  318.731646.563   326.2 1648.14   336.1 1648.69   431.5 1647.93
   459.1 1649.28   478.3 1652.37   504.7 1659.93   521.3  1662.8   543.2 1668.28
   554.3 1670.91   577.5 1678.82     594 1683.41   607.2 1690.73   615.9 1690.55
#Mann= 6 ,-1 , 0
       0      .1       0   17.39      .1       0  213.65     .05       0
  294.83    .045       0  318.73     .05       0   543.2      .1       0
Bank Sta=294.83,318.73
XS Rating Curve= 0 ,0
Exp/Cntr=0.3,0.1

Type RM Length L Ch R = 1 ,7261    ,729.5,731.5,720.9
XS GIS Cut Line= 3
2076425.89539352305489.7154680492076101.24249953305435.896021873
2075792.21490237305394.229110464
#Sta/Elev= 30
       0 1690.96    33.3 1678.02    49.9  1668.2    69.7  1655.2    76.5 1651.84
    92.5 1649.53   103.1 1648.72   163.9 1648.53   206.2 1646.96   235.2 1646.85
  237.851646.103   242.8 1643.56   249.4 1642.91   256.1 1643.72  262.331646.326
   282.7 1646.91   329.2 1646.47   343.9 1646.91   355.7 1646.31   402.1    1647
   418.6  1646.1   445.1 1647.25   505.2 1651.46   574.4 1660.56   608.5 1669.66
   617.3 1673.56   620.6 1675.52   627.2  1680.7   630.5 1682.09   640.9 1681.98
#Mann= 5 ,-1 , 0
       0      .1       0   90.32     .05       0  237.85    .045       0
  262.33     .05       0  587.32      .1       0
Bank Sta=237.85,262.33
XS Rating Curve= 0 ,0
Exp/Cntr=0.3,0.1

Type RM Length L Ch R = 1 ,6529    ,746.4,769.7,748.5
XS GIS Cut Line= 3
2076417.21496469304882.076591462 2076068.2566731304932.423603624
2075790.47868535304946.312683463
#Sta/Elev= 30
       0 1673.11    14.4 1667.88    24.4  1665.3    77.4 1656.17    90.7  1653.4
   109.6 1647.85   130.5 1644.91   140.4 1644.21   176.6 1644.68  186.08 1644.05
   190.1 1642.03   193.4 1641.45   206.7 1641.77  215.461644.595   279.6 1643.91
   306.1 1644.59   332.7 1643.84   395.3 1645.17   424.8    1644   454.4 1645.73
   490.5 1645.28   520.5 1645.94   533.2 1647.64   536.5 1649.05   568.9 1669.23
   598.9 1680.94   604.2 1683.81   615.3 1691.63   618.6 1692.64   630.7 1692.48
#Mann= 7 ,-1 , 0
       0      .1       0    2.21     .05       0   41.22      .1       0
  152.88     .05       0  186.08    .045       0  215.46     .05       0
  557.38      .1       0
#XS Ineff= 2 , 0
                          413.19         1651.83
Permanent Ineff=
       F       F
Bank Sta=186.08,215.46
XS Rating Curve= 0 ,0
Exp/Cntr=0.3,0.1

Type RM Length L Ch R = 1 ,5759    ,846,864.6,844.3
XS GIS Cut Line= 3
2076480.14889395304401.173681885 2076014.0031727304375.132067293
2075726.24259335304364.715421468
#Sta/Elev= 30
       0 1669.81    11.6 1665.14    28.1 1664.76    70.8 1659.23    83.9 1656.38
    93.8  1656.3   139.8 1650.77     150 1648.41   162.4 1644.08   171.7 1642.31
   343.5 1642.82  346.071642.103   350.1 1639.18   356.6 1637.99   361.6 1638.43
  372.191641.873   405.9  1642.8   471.7 1642.33   553.7 1642.99   566.9 1642.91
   586.6 1641.14   632.5 1644.29   658.8 1645.21   671.9 1646.32   688.3 1649.62
     724 1666.64   730.4 1670.21   740.9 1678.42   744.1 1679.78   754.8 1678.75
#Mann= 4 ,-1 , 0
       0     .05       0  346.07    .045       0  372.19     .05       0
     724      .1       0
Bank Sta=346.07,372.19
XS Rating Curve= 0 ,0
Exp/Cntr=0.5,0.3

Type RM Length L Ch R = 1 ,4895    ,44.6,46.4,47.3
XS GIS Cut Line= 3
2076640.54260203303955.328444958 2076213.4591386303964.008873791
2075555.47324985  304026.5087488
#Sta/Elev= 30
       0 1675.83     4.7 1673.21    17.8 1672.06    20.7 1670.84    34.2 1662.92
    50.8 1659.17    73.6 1656.52   126.1 1652.35   162.2 1647.91     195 1645.66
   231.1 1643.95   290.2 1643.36   326.3 1642.05   423.5 1641.43   431.3 1640.22
   441.2 1641.56   467.5 1641.79   490.6 1641.16   610.3 1640.91   619.1 1638.32
   629.8 1638.03   637.4 1638.39   645.5    1641   711.4  1641.6     774 1643.71
   816.9 1647.54   912.5 1650.03  1004.6 1657.35  1057.5 1662.51  1088.1 1666.73
#Mann= 5 ,-1 , 0
       0      .1       0    20.7     .05       0   610.3    .045       0
   645.5     .05       0  1004.6      .1       0
#XS Ineff= 2 , 0
           600.3  1641.4   655.5          1641.4
Permanent Ineff=
       F       F
Bank Sta=610.3,645.5
XS Rating Curve= 0 ,0
Exp/Cntr=0.5,0.3
